HEC-RAS study SMITHCK.prj: SMITHCK

--- SMITHCK.g01 (geometry) --- (continued)

Type RM Length L Ch R = 1 ,37942   ,82.3,74.5,66.7
XS GIS Cut Line= 4
2411681.54799519591423.0834010262411758.28410634591352.250067713
2411852.03410629 591367.180623252411937.10355079591342.875067713
#Sta/Elev= 30
       0 2691.37    16.6    2685      22 2683.43    28.5 2681.01    43.8 2679.67
    49.2 2678.08    53.3 2677.63      71 2677.47    82.3 2676.85    92.8 2675.82
     116 2672.08   128.2 2671.08  148.852668.016   152.5 2666.76   156.5 2665.93
  162.922665.335   168.7    2665  181.252665.356   184.9 2666.46     193 2669.98
   201.4 2670.59   213.6 2670.55   226.1 2670.04   234.4 2668.68   238.5 2668.59
   246.9 2670.44  251.072672.338   267.7 2682.02   278.6 2689.04   287.8 2695.48
#Mann= 5 ,-1 , 0
       0      .1       0  148.85     .06       0  162.92    .045       0
  181.25     .06       0  251.07      .1       0
#XS Ineff= 2 , 0
                          209.36         2669.83
Permanent Ineff=
       F       F
Bank Sta=162.92,181.25
XS Rating Curve= 0 ,0
Exp/Cntr(USF)=0,0
Exp/Cntr=0.5,0.3

Type RM Length L Ch R = 1 ,37867   ,66.6,75.3,80.1
XS GIS Cut Line= 2
2411738.37658275591482.3460543262411947.35682199591388.772812872
#Sta/Elev= 30
       0 2674.52    12.4 2672.48    23.3 2671.19    29.3  2671.1    50.5 2671.67
      65  2671.6    73.8 2671.31   85.542670.377    91.3 2669.62    95.7 2668.46
      99 2667.03     105 2663.21   108.8 2661.53  111.092661.102   117.1 2660.63
     122 2660.81  123.192661.078   126.4 2661.91   135.1 2666.23   138.3 2666.87
     157 2667.23   170.2 2666.71   174.6 2666.25     179 2666.45   183.3 2667.96
  188.312670.351   192.1 2672.47   200.9 2678.55   207.9 2682.69     229 2692.29
#Mann= 5 ,-1 , 0
       0      .1       0   85.54     .06       0  111.09    .045       0
  123.19     .06       0  188.31      .1       0
#XS Ineff= 2 , 0
                          150.79         2668.36
Permanent Ineff=
       F       F
Bank Sta=111.09,123.19
XS Rating Curve= 0 ,0
Exp/Cntr(USF)=0,0
Exp/Cntr=0.3,0.1

Type RM Length L Ch R = 1 ,37792   ,115.4,118.1,117
XS GIS Cut Line= 2
2411747.73979885591491.9150858082411987.91111858591516.867950196
#Sta/Elev= 30
       0 2672.94    14.1  2670.4    18.1 2669.95    25.8 2669.58    46.2 2669.23
    62.3 2668.48    74.4 2667.71   77.642667.304    90.5 2665.44    94.5 2664.46
   106.5  2660.5  110.582659.346   114.6 2658.71   122.6 2658.52   126.6 2658.94
  127.412659.291   134.7 2663.18   138.7 2663.66   150.8 2663.34   154.8  2663.9
   170.9 2670.61   174.9 2672.76  180.532676.428   186.7 2680.95   207.1 2697.13
   219.1 2705.52   223.1 2707.85   227.7 2709.78   235.2 2712.32   241.5 2713.78
#Mann= 5 ,-1 , 0
       0      .1       0   77.64     .06       0  110.58    .045       0
  127.41     .06       0  180.53      .1       0
#XS Ineff= 2 , 0
                          138.94         2667.71
Permanent Ineff=
       F       F
Bank Sta=110.58,127.41
XS Rating Curve= 0 ,0
Exp/Cntr(USF)=0,0
Exp/Cntr=0.3,0.1

Type RM Length L Ch R = 1 ,37674   ,140.8,140.4,139.9
XS GIS Cut Line= 2
2411753.97801494591597.9647594552411959.83914614 591629.15583994
#Sta/Elev= 30
       0 2671.23     7.8 2667.44    11.9 2665.86      20 2663.87      24 2663.18
    28.1 2663.01    36.1 2663.21    40.2 2662.85    44.2  2660.1    48.3 2656.27
    52.3 2653.58      552653.027    56.8 2652.73   70.712652.977    76.6 2653.28
    84.7 2655.45   90.092656.027    92.8    2656   100.9 2656.66     113 2658.12
   121.1 2657.66   137.3 2657.69   141.1 2660.28   145.4  2663.6   148.1 2665.35
   177.7  2682.1   185.8 2687.73  194.412693.183   198.8 2695.58   208.2 2699.75
#Mann= 5 ,-1 , 0
       0      .1       0      55    .045       0   70.71      .1       0
   90.09     .06       0  194.41      .1       0
#XS Ineff= 2 , 0
                          112.74          2658.5
Permanent Ineff=
       F       F
Bank Sta=55,70.71
XS Rating Curve= 0 ,0
Exp/Cntr(USF)=0,0
Exp/Cntr=0.3,0.1

Type RM Length L Ch R = 1 ,37534   ,143.7,143.6,143.2
XS GIS Cut Line= 3
2411704.07228617591735.2055135872411891.21876907591753.920161878
2411981.67290248591722.729081393
#Sta/Elev= 30
       0 2676.13    37.8 2663.11    49.9 2658.15   59.692655.401      66 2654.48
      74 2654.13      78 2652.73   85.292646.937    86.1 2646.36    90.1 2645.59
    94.1 2645.57  100.492646.779   106.2 2647.23   118.1 2651.13   122.2 2651.79
   146.4 2652.28   158.4 2651.87  162.472652.809   166.5 2654.64   170.5 2655.76
   186.6 2655.14   190.7 2655.66   194.9 2656.74   199.2 2658.33   220.7 2668.27
     233 2672.93   245.7 2679.97   249.9 2681.94   258.4 2685.42   283.8 2694.61
#Mann= 5 ,-1 , 0
       0      .1       0   59.69     .06       0   85.29    .045       0
  100.49     .06       0  162.47      .1       0
#XS Ineff= 2 , 0
                          130.61          2656.5
Permanent Ineff=
       F       F
Bank Sta=85.29,100.49
XS Rating Curve= 0 ,0
Exp/Cntr(USF)=0,0
Exp/Cntr=0.3,0.1

Type RM Length L Ch R = 1 ,37390   ,123.8,120,114.4
XS GIS Cut Line= 2
2411689.89247441591878.7695661522411956.74949634591899.563619808
#Sta/Elev= 30
       0 2663.13     8.4 2658.16    15.9 2654.57    19.9 2653.13    23.9  2652.3
    39.9 2650.41      44  2649.5      56 2645.63      60 2644.55      64 2643.86
    89.3 2642.74    92.1 2642.47   97.412641.263  103.332640.312   108.1 2639.84
  116.192640.309   126.5 2641.85   136.2 2642.06   148.3 2643.29   152.3 2644.43
   156.2 2646.61   160.3 2648.53   164.3 2648.73   172.3 2648.32  199.622647.948
   228.5 2647.66   236.5 2648.28   252.6 2652.49   260.8    2655   267.7 2657.64
#Mann= 5 ,-1 , 0
       0      .1       0   97.41     .06       0  103.33    .045       0
  116.19     .06       0  199.62      .1       0
Bank Sta=103.33,116.19
XS Rating Curve= 0 ,0
Exp/Cntr(USF)=0,0
Exp/Cntr=0.3,0.1

Type RM Length L Ch R = 1 ,37270   ,131.9,131.3,126.7
XS GIS Cut Line= 2
2411736.19566805592019.6397837232411955.16547464591958.246380005
#Sta/Elev= 30
       0 2651.85     5.7 2647.42     9.9 2644.55      14  2642.2    18.2 2640.37
    22.4 2639.42    26.5 2639.03    34.8 2639.61    37.6 2639.32      39  2639.1
    43.1 2637.38    47.3 2636.34    55.42635.932    63.5  2635.5    73.2 2635.85
    86.2 2637.28   105.4 2635.66   109.6 2636.68     122 2642.41   126.2 2643.15
   134.5 2643.34     147 2643.01   151.1 2643.53   155.3 2644.94   159.4 2645.68
   171.9 2645.23     190 2643.21   205.1 2643.49   221.7 2646.59   227.4 2648.84
#Mann= 4 ,-1 , 0
       0      .1       0    55.4    .045       0    73.2     .06       0
   171.9      .1       0
Bank Sta=55.4,73.2
XS Rating Curve= 0 ,0
Exp/Cntr(USF)=0,0
Exp/Cntr=0.3,0.1

Type RM Length L Ch R = 1 ,37139   ,116.8,121.7,124.9
XS GIS Cut Line= 2
2411734.94625733592145.6265880752412005.26895487592048.587671012
#Sta/Elev= 30
       0 2664.82    15.7 2655.93    26.2 2649.18    36.9 2642.94    49.7 2637.22
    63.8 2637.65    83.7 2632.28    87.9 2631.76   94.482631.791   113.4 2632.65
   126.2    2629   135.7 2630.22   151.3 2630.59  158.512627.728   164.4 2626.85
   168.7 2627.18  170.112627.787   177.2 2632.96   181.4 2633.82  195.512634.004
   198.4 2634.39   202.7 2635.78   215.4 2641.52   219.7 2642.54   229.5 2643.63
   249.4 2647.39   262.2 2652.81   270.7  2655.2   279.5 2660.57   287.2 2664.57
#Mann= 5 ,-1 , 0
       0      .1       0   94.48     .06       0  158.51    .045       0
  170.11     .06       0  195.51      .1       0
#XS Ineff= 2 , 0
           110.1 2632.83
Permanent Ineff=
       F       F
Bank Sta=158.51,170.11
XS Rating Curve= 0 ,0
Exp/Cntr(USF)=0,0
Exp/Cntr=0.3,0.1

Type RM Length L Ch R = 1 ,37017   ,119.8,113.6,106.3
XS GIS Cut Line= 3
2411766.89236991592201.7735480852411965.39770859592209.959335247
2412039.06979306592179.262633389
#Sta/Elev= 30
       0 2658.53    19.1 2645.88    26.8 2640.13    38.3 2630.67    42.9 2628.06
    46.9 2627.23    71.82627.385    82.9 2628.01    86.9 2627.32    94.9 2622.21
   97.892621.801   102.9 2621.29  111.392621.638   122.9 2624.34   146.9 2628.59
   150.9  2628.2   158.9 2626.35     171 2626.05     175 2626.93     183 2629.88
     191 2631.54   203.3 2635.29   207.7 2636.02   220.7  2636.6   229.3 2637.96
     238 2641.34     251 2647.94   259.4 2652.86   275.1 2660.12   278.5 2661.81
#Mann= 5 ,-1 , 0
       0      .1       0    71.8     .06       0   97.89    .045       0
  111.39     .06       0   275.1      .1       0
#XS Ineff= 2 , 0
                          149.24         2627.09
Permanent Ineff=
       F       F
Bank Sta=97.89,111.39
XS Rating Curve= 0 ,0
Exp/Cntr(USF)=0,0
Exp/Cntr=0.3,0.1

Type RM Length L Ch R = 1 ,36903   ,151.9,155.5,159.3
XS GIS Cut Line= 2
2411821.58814757592357.0328002482412039.92571096592235.734153919
#Sta/Elev= 30
       0 2663.55    18.4 2652.03    22.3 2649.12    27.6  2644.3    31.1 2642.85
      37 2641.22    50.5 2631.39    59.6 2625.75    70.5 2621.76    77.9 2618.55
   84.092617.481    98.8 2617.23  101.692617.398   105.4 2618.26   114.5 2621.96
   116.4 2622.19   119.4 2622.28   128.2 2620.69   137.4 2620.34     140 2620.67
     142 2621.08  149.392624.993   152.8 2625.93   164.9    2626   169.4 2626.81
   183.2 2630.64   196.9 2632.87   204.7  2634.8   219.8  2640.3   249.8 2653.49
#Mann= 4 ,-1 , 0
       0      .1       0   84.09    .045       0  101.69      .1       0
  149.39     .06       0
#XS Ineff= 2 , 0
                          118.63         2621.94
Permanent Ineff=
       F       F
Bank Sta=84.09,101.69
XS Rating Curve= 0 ,0
Exp/Cntr(USF)=0,0
Exp/Cntr=0.3,0.1

Type RM Length L Ch R = 1 ,36748   ,149.8,153.3,155.8
XS GIS Cut Line= 2
2411845.84787683592481.797122186 2412126.5676012592412.483609998
#Sta/Elev= 30
       0 2662.09    24.6 2646.07    32.8 2643.27    48.6 2632.29    65.1 2623.21
      74 2619.01    82.2 2615.98    86.4 2615.38    94.9 2615.48    98.7 2614.55
   102.8 2612.34  105.082611.844   119.3 2611.09  124.782611.542     1372612.704
   164.6 2613.09   177.5 2613.85   185.2 2615.44   189.4 2615.19   193.5 2613.89
   197.3  2613.4   207.2 2613.36   210.5 2614.34   226.4 2624.12  236.652631.221
   255.3 2643.86   266.7 2650.75   275.9 2658.14   283.2  2663.1   289.2 2668.31
#Mann= 5 ,-1 , 0
       0      .1       0  105.08    .045       0  124.78      .1       0
     137     .06       0  236.65      .1       0
#XS Ineff= 2 , 0
                          186.71         2615.53
Permanent Ineff=
       F       F
Bank Sta=105.08,124.78
XS Rating Curve= 0 ,0
Exp/Cntr(USF)=0,0
Exp/Cntr=0.3,0.1

Type RM Length L Ch R = 1 ,36594   ,100.3,97.8,96.7
XS GIS Cut Line= 3
2411845.84787683592589.2330660772412081.51381827592596.164417296
2412192.41543777592537.247931936
#Sta/Elev= 30
       0 2666.86     7.9 2660.55    19.9 2656.64    31.2 2647.78    59.9 2629.53
    76.6 2621.55    91.9  2615.1   111.9 2608.67   119.9 2608.04   131.9 2604.46
  150.922601.138   159.9 2600.67  164.622601.004   167.9 2601.72   175.9 2607.07
   179.9 2608.76   184.1 2609.36   211.9 2607.75   258.6  2608.3   272.2 2606.79
   285.8 2606.61   289.9 2608.52   294.8 2613.08     313 2626.19   326.5 2639.25
   335.6 2646.63   344.7 2653.19   349.5 2658.57   353.7  2661.5   361.3 2665.35
#Mann= 3 ,-1 , 0
       0      .1       0  150.92    .045       0  164.62     .06       0
Bank Sta=150.92,164.62
XS Rating Curve= 0 ,0
Exp/Cntr(USF)=0,0
Exp/Cntr=0.3,0.1

Type RM Length L Ch R = 1 ,36497   ,124.7,117.9,113.6
XS GIS Cut Line= 3
  2411858.354757592701.8901808732412158.72486207592673.818208437
2412242.94077938592628.903052539
#Sta/Elev= 30
       0 2659.52     7.4 2657.28    15.4 2653.44    39.5 2639.43    71.7 2624.17
    99.8 2606.52   103.8 2604.62   112.5  2602.3   119.8  2598.3  122.342597.637
   127.9 2597.06  139.912597.622   168.1 2605.36   216.3 2601.63   228.3 2603.27
   240.4 2603.78  259.342601.435   268.5 2600.76   276.5 2601.89   284.6 2601.63
   296.6 2604.84   309.6 2603.81   318.6 2609.17   341.6 2619.99   353.4 2627.53
  361.992631.199     380 2638.74   386.6 2642.47   391.1 2643.88   397.1 2644.53
#Mann= 5 ,-1 , 0
       0      .1       0  122.34    .045       0  139.91      .1       0
  259.34     .06       0  361.99      .1       0
#XS Ineff= 2 , 0
                          189.85          2603.3
Permanent Ineff=
       F       F
Bank Sta=122.34,139.91
XS Rating Curve= 0 ,0
Exp/Cntr(USF)=0,0
Exp/Cntr=0.3,0.1

Type RM Length L Ch R = 1 ,36379   ,187.1,187.6,188.3
XS GIS Cut Line= 2
2411960.21517194592831.8303587342412247.86624752592672.409280702
#Sta/Elev= 30
       0 2621.25    24.6 2609.56    40.1 2604.11    47.4 2602.75    56.6  2603.5
    60.7 2603.08    65.7 2601.03    70.3 2598.24    74.9 2596.59    88.6 2595.07
    97.7 2592.19  101.192591.891   111.4 2591.43  116.932591.786   119.6 2592.87
     126 2597.22   157.2  2600.5   167.2 2600.46   181.3 2597.67  190.232597.364
   202.9 2599.28   207.5 2600.53   216.6 2604.19   221.2 2605.17   231.4 2605.73
   248.6  2605.6   257.8 2610.07   276.1  2613.5  295.782618.429   328.9 2625.71
#Mann= 5 ,-1 , 0
       0      .1       0  101.19    .045       0  116.93      .1       0
  190.23     .06       0  295.78      .1       0
Bank Sta=101.19,116.93
XS Rating Curve= 0 ,0
Exp/Cntr(USF)=0,0
Exp/Cntr=0.3,0.1

Type RM Length L Ch R = 1 ,36191   ,131.2,132.9,132.6
XS GIS Cut Line= 2
2412026.06300852592994.7171123752412365.69921824592828.364683125
#Sta/Elev= 30
       0 2615.69    35.2 2598.33    54.5 2591.22    61.9 2590.61    97.6 2591.86
   106.5 2590.39   119.8  2586.1   124.3 2585.57   142.1 2586.26  146.382584.876
     151 2583.73   159.9 2583.45  165.092583.808   168.8 2584.65   177.7 2590.87
   182.2 2591.86     203 2590.82   213.4 2594.42   240.1 2594.98     249 2596.94
   257.9 2601.03   265.8 2605.73   283.7 2618.19   289.1 2622.55   302.4 2636.45
  308.932642.061   315.8 2646.36   329.1 2653.19   355.4 2664.54   378.2 2673.25
#Mann= 5 ,-1 , 0
       0      .1       0  146.38     .06       0     151    .045       0
  165.09     .06       0  308.93      .1       0
Bank Sta=151,165.09
XS Rating Curve= 0 ,0
Exp/Cntr(USF)=0,0
Exp/Cntr=0.3,0.1

Type RM Length L Ch R = 1 ,36058   ,111,112.2,111.2
XS GIS Cut Line= 2
 2412057.6657613593108.9337811972412416.98700848592957.345130042
#Sta/Elev= 30
       0 2617.45      13 2612.82    35.3 2607.81    69.5 2598.41    95.5 2593.24
   112.9 2588.42   121.6 2585.15   138.9  2582.6   146.1 2579.18     152  2578.6
   160.6 2578.97   173.7 2581.13   186.7 2585.93   195.4 2587.27     204 2587.44
   217.1  2585.7  233.072585.025   238.8 2584.75   247.5 2582.94   260.5 2583.12
   264.8 2584.01   269.2 2585.92   288.7 2597.91   308.2 2611.31   312.6 2615.15
   325.6 2629.35  335.282637.143   343.6 2642.75   360.3 2652.24     390 2666.48
#Mann= 5 ,-1 , 0
       0      .1       0   146.1    .045       0   160.6      .1       0
  233.07     .06       0  335.28      .1       0
#XS Ineff= 2 , 0
                          196.62         2587.84
Permanent Ineff=
       F       F
Bank Sta=146.1,160.6
XS Rating Curve= 0 ,0
Exp/Cntr(USF)=0,0
Exp/Cntr=0.3,0.1

Type RM Length L Ch R = 1 ,35946   ,219,218.2,217.9
XS GIS Cut Line= 2
2412112.70489876593192.2606221112412476.60083774593060.564948954
#Sta/Elev= 30
       0 2616.89     9.5 2614.04    43.6 2606.99    60.6 2602.63    86.1 2593.13
   103.1 2590.69   115.9 2587.82   124.4 2584.32   137.1  2577.2   141.4 2575.79
   149.9 2574.54   156.42574.568   164.4 2574.29   167.5 2574.42   176.9 2580.22
  188.762580.897   213.7 2580.21   226.5 2580.93     235 2579.43     252 2579.04
   264.7 2585.37   273.3 2590.85  289.83 2602.97   298.7  2609.4   307.3 2619.69
   311.5 2623.59   328.5 2636.85   358.3 2655.84   366.8 2660.54     387    2670
#Mann= 5 ,-1 , 0
       0      .1       0   156.4    .045       0   167.5      .1       0
  188.76     .06       0  289.83      .1       0
#XS Ineff= 2 , 0
                          183.99         2583.76
Permanent Ineff=
       F       F
Bank Sta=156.4,167.5
XS Rating Curve= 0 ,0
Exp/Cntr(USF)=0,0
Exp/Cntr=0.3,0.1

Type RM Length L Ch R = 1 ,35728   ,274.1,267.1,263.5
XS GIS Cut Line= 2
2412188.94976216593396.735483065 2412608.2965109593237.314405033
#Sta/Elev= 30
       0  2610.6    43.6 2594.78    82.1 2583.69   103.5 2575.09     112 2570.65
  127.462567.148   146.3 2566.78  147.812567.073   150.5 2567.79   159.1 2573.22
   163.4 2573.88   184.8 2572.66   197.6 2569.69   201.9 2569.38   228.5 2569.52
  247.322571.216   278.9  2570.1   283.2 2570.59   291.7 2575.05   299.8 2577.37
   304.6 2579.95   318.4 2588.74   334.5 2601.55  348.722609.963   364.5 2618.78
   386.6 2629.83   411.5 2640.32   420.1 2642.09   426.9 2642.33   448.6 2639.16
#Mann= 5 ,-1 , 0
       0      .1       0  127.46    .045       0  147.81      .1       0
  247.32     .06       0  348.72      .1       0
#XS Ineff= 2 , 0
                          165.16          2574.6
Permanent Ineff=
       F       F
Bank Sta=127.46,147.81
XS Rating Curve= 0 ,0
Exp/Cntr(USF)=0,0
Exp/Cntr=0.3,0.1

Type RM Length L Ch R = 1 ,35461   ,84.1,79.9,74
XS GIS Cut Line= 2
2412337.97381337593667.0581805972412688.00704992593351.681700143
#Sta/Elev= 30
       0 2620.22    21.1 2612.54    48.2 2600.54    54.4 2598.61    85.7 2582.82
     119 2568.56   134.2 2560.44   139.5    2559   147.3 2558.49   155.7 2558.49
   167.9 2559.91  180.082556.234     188 2555.42  197.782556.266   204.1 2559.51
   209.6 2560.84  221.492560.233   251.5 2558.88   279.5 2559.17   283.2 2559.82
   305.9 2569.11   320.1  2577.6   333.3 2588.15   341.2 2592.16   360.3 2599.41
   381.8 2603.87  399.672606.365   430.3 2609.27   435.6 2609.02   471.2  2613.1
#Mann= 5 ,-1 , 0
       0      .1       0  180.08    .045       0  197.78      .1       0
  221.49     .06       0  399.67      .1       0
#XS Ineff= 2 , 0
                          209.99         2563.75
Permanent Ineff=
       F       F
Bank Sta=180.08,197.78
XS Rating Curve= 0 ,0
Exp/Cntr(USF)=0,0
Exp/Cntr=0.5,0.3

Type RM Length L Ch R = 1 ,35381   ,40.7,41.1,41.8
XS GIS Cut Line= 4
2412365.31535639593743.6563177112412500.73202294593662.493123263
2412568.44035634593466.7465954722412699.95077296593348.257012144
#Sta/Elev= 30
       0 2619.16    25.3 2611.65    64.2  2597.3   112.3 2576.62   134.2 2568.13
   154.3 2554.73     171 2553.24   183.1 2553.17   195.8  2556.3   204.2 2555.26
  209.612553.318   216.9 2552.68  221.81 2552.87   237.1 2553.33   246.7 2556.13
   276.2  2557.7  318.252557.696   331.9 2557.55     344 2559.94   368.7 2570.71
   377.4 2575.92   393.5 2587.09   415.1 2597.19   420.4 2599.16   436.6 2602.82
  457.23 2605.93   478.6 2608.03   493.3 2608.32   517.3 2610.89     542 2615.27
#Mann= 5 ,-1 , 0
       0      .1       0  209.61    .045       0  221.81      .1       0
  318.25     .06       0  457.23      .1       0
#XS Ineff= 2 , 0
                          250.96         2561.76
Permanent Ineff=
       F       F
Bank Sta=209.61,221.81
XS Rating Curve= 0 ,0
Exp/Cntr(USF)=0,0
Exp/Cntr=0.5,0.3

Type RM Length L Ch R = 1 ,35340   ,107.6,112.3,114.2
XS GIS Cut Line= 4
2412401.33966194593763.187567711 2412536.7563285593682.024373263
 2412604.4646619593486.2778454722412735.97507851593367.788262144
#Sta/Elev= 30
       0 2600.26    28.3 2589.99    56.3 2578.48   102.9 2562.61   112.3 2560.33
   135.6 2556.68   144.9 2553.83   157.9 2552.96   169.9 2549.89   174.1 2549.61
   191.1 2552.98  213.612551.379  229.112551.461   246.1 2551.94  250.562553.504
   254.5 2555.14   258.7 2555.56   313.8 2554.87   322.2 2555.98     331 2559.19
   347.6 2569.14   356.1 2573.13   370.4    2578   398.9 2590.85  418.64 2596.15
   441.9 2600.85   458.1 2600.77   477.9 2603.21   512.8 2608.98     542  2611.7
#Mann= 5 ,-1 , 0
       0      .1       0  213.61    .045       0  229.11      .1       0
  250.56     .06       0  418.64      .1       0
#XS Ineff= 4 ,-1
       0   202.5    2553   237.5  260.43    2553  260.43  371.36 2559.68
  371.36     542    2553
Permanent Ineff=
       F       F       F       F
Bank Sta=213.61,229.11
XS Rating Curve= 0 ,0
Exp/Cntr(USF)=0,0
Exp/Cntr=0.5,0.3

Type RM Length L Ch R = 1 ,35227   ,116.8,118.6,119.8
XS GIS Cut Line= 3
2412532.05164753593850.7389879082412708.80110358 593576.95061475
2412735.54105078593372.996595472
#Sta/Elev= 30
       0 2591.68    12.8 2591.56    33.4 2588.08    47.2 2582.59      81 2563.72
   100.1 2557.81   114.4 2551.39   138.2 2547.58   150.4 2544.18   157.2 2544.87
   171.9  2547.7  184.072548.256     202 2549.07   219.1    2549   228.6 2547.89
  235.492545.713   238.4 2545.04   247.1 2544.78  252.392546.057   261.9 2550.23
     300 2550.21   304.8 2552.22  314.642557.785   328.6 2565.42   348.3 2572.55
   428.5 2591.25   446.3 2593.29   481.5 2600.15   509.7 2606.79   531.6 2610.77
#Mann= 5 ,-1 , 0
       0      .1       0  184.07     .06       0  235.49    .045       0
  252.39     .06       0  314.64      .1       0
Bank Sta=235.49,252.39
XS Rating Curve= 0 ,0
Exp/Cntr(USF)=0,0
Exp/Cntr=0.3,0.1

Type RM Length L Ch R = 1 ,35109   ,131.4,131.6,130.3
XS GIS Cut Line= 3
2412621.91240726593880.913023189 2412824.0306088593636.686862995
2412840.87379227593423.339872481
#Sta/Elev= 30
       0 2615.88     7.1 2612.38    44.5  2590.8   117.2  2541.4   122.3 2540.13
  125.972540.772   132.7 2543.58   137.6 2543.87   181.5 2544.16  189.812541.947
     195    2541  206.612541.752   220.1 2546.04   225.4 2546.84  252.892544.874
   285.5 2542.91   293.7 2543.22   304.1 2545.16   314.4 2545.32     319 2546.56
   327.1 2553.24   338.9 2560.19   347.1 2562.63   367.2 2567.03  387.242572.254
   395.3 2573.14   427.4 2580.81   448.2 2584.38   479.5 2591.41     531 2599.77
#Mann= 6 ,-1 , 0
       0      .1       0  125.97      .1       0  189.81    .045       0
  206.61      .1       0  252.89     .06       0  387.24      .1       0
#XS Ineff= 2 , 0
                          226.07         2552.34
Permanent Ineff=
       F       F
Bank Sta=189.81,206.61
XS Rating Curve= 0 ,0
Exp/Cntr(USF)=0,0
Exp/Cntr=0.3,0.1

Type RM Length L Ch R = 1 ,34977   ,94.5,97.4,98.2
XS GIS Cut Line= 3
2412712.26677918 593989.366012272412930.60434257593698.249261081
2412909.81028892593452.186292815
#Sta/Elev= 30
       0  2631.5    15.6 2623.77    34.3  2612.9    53.4 2603.84   108.6 2580.91
   151.5 2566.64  164.532561.024   185.7 2546.81  197.212536.494   198.4  2535.8
   203.4 2535.38  214.31 2536.18   228.9 2537.89   248.4  2537.8   254.3 2539.19
     260 2539.69   282.2 2539.51  292.972538.096   322.9 2537.72   334.3 2539.91
   348.4 2540.21   362.2 2545.31   388.6 2550.45  412.012553.876   447.8 2562.16
   487.9 2569.06   532.1 2578.12   576.2 2584.73  607.542590.605   610.8 2591.33
#Mann= 7 ,-1 , 0
       0      .1       0  164.53      .1       0  197.21    .045       0
  214.31      .1       0  292.97     .06       0  412.01      .1       0
  607.54      .1       0
#XS Ineff= 2 , 0
                          268.35         2547.48
Permanent Ineff=
       F       F
Bank Sta=197.21,214.31
XS Rating Curve= 0 ,0
Exp/Cntr(USF)=0,0
Exp/Cntr=0.3,0.1

Type RM Length L Ch R = 1 ,34880   ,131.4,133.1,134.4
XS GIS Cut Line= 2
2412767.88666393 594021.272885372413149.66548906593633.879665751
#Sta/Elev= 30
       0 2611.17    14.9 2601.21    34.2 2591.98    54.2 2583.54   85.16 2572.68
   104.9 2565.58   138.5 2551.98   150.6 2546.37     162 2539.66   169.9 2536.03
   179.1 2534.36   201.9 2534.31   209.5 2532.38     218 2531.03   226.5 2532.38
   229.3 2533.34     235  2536.7  246.872535.781   267.6 2533.39   290.1 2532.53
   312.6 2533.04   325.5 2534.83   355.7 2533.51   372.8 2534.13   389.9 2537.31
   402.4 2541.86  410.512543.966  454.43 2547.57   509.1 2552.69   543.9 2558.91
#Mann= 7 ,-1 , 0
       0      .1       0   85.16      .1       0   209.5    .045       0
   226.5      .1       0  246.87     .06       0  410.51      .1       0
  454.43      .1       0
#XS Ineff= 2 , 0
                          239.87         2543.81
Permanent Ineff=
       F       F
Bank Sta=209.5,226.5
XS Rating Curve= 0 ,0
Exp/Cntr(USF)=0,0
Exp/Cntr=0.3,0.1

Type RM Length L Ch R = 1 ,34747   ,278.5,276.6,276.2
XS GIS Cut Line= 3
2412812.77137185594117.5960098182413041.50596207593937.380878129
2413263.30920108593691.317909863
#Sta/Elev= 30
       0 2615.16   45.552591.453    77.4 2575.65    99.5 2568.14   134.1 2560.26
   156.5 2552.54   173.6 2543.21   187.8 2531.82   192.2  2529.3   196.4 2528.53
   207.8 2529.24  214.892527.124   230.2  2526.5  235.292527.427   240.4 2529.46
   250.6 2529.83   260.7 2531.91  305.032531.685   355.5 2526.46     369 2525.99
   386.6 2528.23   417.8 2527.85   434.8 2535.86  459.552537.639   500.4  2538.3
   519.7 2540.39   560.1 2550.91   579.2 2553.34   607.2 2565.45   622.5 2568.91
#Mann= 6 ,-1 , 0
       0      .1       0   45.55      .1       0  214.89    .045       0
  235.29      .1       0  305.03     .06       0  459.55      .1       0
#XS Ineff= 2 , 0
                          284.45         2539.05
Permanent Ineff=
       F       F
Bank Sta=214.89,235.29
XS Rating Curve= 0 ,0
Exp/Cntr(USF)=0,0
Exp/Cntr=0.3,0.1

Type RM Length L Ch R = 1 ,34470   ,189.9,192.6,194
XS GIS Cut Line= 3
2412850.89380356594280.4827634592413193.99568889 594103.73330738
2413440.05865715593829.944934238
#Sta/Elev= 30
       0 2623.81    43.5  2605.6   108.9  2581.5   117.6 2576.94   134.1 2573.77
   160.5 2561.92   241.5 2532.86     246 2532.39     255 2533.39   277.5 2529.93
     318 2528.62   349.5 2525.29   414.8 2522.85   426.1 2521.44  435.782517.577
   448.7 2516.27  459.582517.742  461.162518.521   469.1 2524.64   475.1 2527.66
   500.4 2528.39   513.9 2530.99   528.9 2532.05   550.7 2536.84  588.672543.035
     613 2546.92   629.4  2551.6   672.5 2557.59   710.1  2565.4   754.1 2577.72
#Mann= 5 ,-1 , 0
       0      .1       0  435.78    .045       0  459.58      .1       0
  461.16     .06       0  588.67      .1       0
Bank Sta=435.78,459.58
XS Rating Curve= 0 ,0
Exp/Cntr(USF)=0,0
Exp/Cntr=0.3,0.1

Type RM Length L Ch R = 1 ,34278   ,84.7,86.1,87
XS GIS Cut Line= 3
     2413051.006      594466.854 2413423.3271878594143.684217078
2413499.17751709593897.907217078
#Sta/Elev= 30
       0 2587.26    45.8 2569.58   110.2 2542.79   146.8  2531.5   177.8  2523.6
     214 2519.75   231.1 2512.46   237.3 2511.45   268.9 2512.37   323.8 2510.69
   339.4  2511.6   358.2 2509.83   379.1 2511.34  398.912502.038   407.4 2501.38
  418.822502.225     420 2502.52   432.4 2508.21     450 2509.42   464.1 2518.28
   469.5 2520.03   533.7 2524.71   544.4 2526.71  576.852536.131   611.3  2545.8
   628.1 2546.92   649.2 2551.06   681.1 2561.56   720.2 2572.09   750.2 2582.96
#Mann= 5 ,-1 , 0
       0      .1       0  398.91    .045       0  418.82      .1       0
     420     .06       0  576.85      .1       0
Bank Sta=398.91,418.82
XS Rating Curve= 0 ,0
Exp/Cntr(USF)=0,0
Exp/Cntr=0.5,0.3

Type RM Length L Ch R = 1 ,34191   ,41.2,41.3,41.2
XS GIS Cut Line= 3
2413092.31188408  594503.20492882413459.49938411 594231.50353992
2413515.48896742593923.343817711
#Sta/Elev= 30
       0 2586.79    56.3 2562.77    91.1  2549.7   147.2 2528.99   180.7 2519.81
   185.7 2517.49   190.6 2512.66     196 2509.66   258.7 2506.26   338.8 2507.17
  362.552504.616   375.9 2503.53  385.692499.313   390.2 2498.34   397.8 2498.17
   404.6 2498.57  407.092499.845     416    2505   438.9 2506.67   449.4 2510.27
   482.1 2512.23  503.422512.116   521.2 2512.62   535.3 2514.21   576.3 2522.76
   648.5  2544.1   688.8 2557.79   717.3 2566.53   738.5 2572.18     770 2577.94
#Mann= 5 ,-1 , 0
       0      .1       0  362.55     .06       0  385.69    .045       0
  407.09     .06       0  503.42      .1       0
#XS Ineff= 2 , 0
             370    2503     420            2503
Permanent Ineff=
       F       F
Bank Sta=385.69,407.09
XS Rating Curve= 0 ,0
Exp/Cntr(USF)=0,0
Exp/Cntr=0.5,0.3

Type RM Length L Ch R = 1 ,34150   ,74.9,72,69.4
XS GIS Cut Line= 3
2413115.74938408594537.0590954672413482.93688411594265.357706587
2413538.92646742593957.197984378
#Sta/Elev= 30
       0    2594    37.4 2575.84     106 2545.45   128.9 2536.43   176.4 2522.08
   186.4 2517.44   196.3 2511.48   199.2 2510.58   206.1 2509.19   226.1 2508.44
     251 2505.29  342.622503.087     372 2503.75   375.4 2503.14  387.392498.443
   397.7 2496.82   405.3 2497.03  409.092498.146   417.7 2504.19   423.4 2506.07
  467.872508.051   532.7 2509.32     549 2510.74   574.9 2515.84     610  2524.8
   634.4 2529.74     671  2541.6   719.4 2560.99   748.2  2573.5     770 2581.07
#Mann= 5 ,-1 , 0
       0      .1       0  342.62     .06       0  387.39    .045       0
  409.09     .06       0  467.87      .1       0
#XS Ineff= 2 , 0
          370.42 2504.17
Permanent Ineff=
       F       F
Bank Sta=387.39,409.09
XS Rating Curve= 0 ,0
Exp/Cntr(USF)=0,0
Exp/Cntr=0.5,0.3

Type RM Length L Ch R = 1 ,34078   ,251.1,246.3,246.4
XS GIS Cut Line= 3
2413203.62648536594645.4661609692413550.96027666594283.948439069
2413593.73535367593945.197919516
#Sta/Elev= 30
       0 2603.59    54.3 2580.24   113.7 2549.72   135.6 2540.38   153.3 2534.47
     176  2529.5   184.5 2525.86   198.1 2524.91   204.3 2523.29   253.6 2505.98
   323.1 2501.75   343.4 2497.84   375.6 2498.55  392.292495.302   408.9 2494.51
  416.392495.268   425.5 2496.77   436.6 2502.24   441.5 2502.87   458.8    2502
   475.5 2504.67   498.4  2503.5  542.22 2503.69   595.4 2504.97  618.192509.685
  643.692513.682     668 2519.49   712.2 2537.56   792.9 2576.81   842.8 2596.93
#Mann= 6 ,-1 , 0
       0      .1       0  392.29    .045       0  416.39     .06       0
  542.22      .1       0  618.19      .1       0  643.69      .1       0
Bank Sta=392.29,416.39
XS Rating Curve= 0 ,0
Exp/Cntr(USF)=0,0
Exp/Cntr=0.3,0.1

Type RM Length L Ch R = 1 ,33832   ,205.4,205.2,205.8
XS GIS Cut Line= 2
     2413436.317      594780.568     2413961.158      594107.777
#Sta/Elev= 30
       0 2550.46    22.9  2552.3    48.2 2551.58    88.8 2544.47   138.5 2540.71
   210.5  2532.5   216.6 2530.32   251.1 2507.51   291.7 2487.64     312 2485.58
   327.2 2490.25   403.3 2488.27   418.5 2491.05   428.7 2490.12  441.092486.464
   450.7 2484.39  461.092486.514   469.6 2492.84   478.2 2494.22   550.4 2490.56
  578.572491.051  605.972491.294   666.3 2490.93   691.9 2492.68     7142497.323
  748.412511.294   801.8 2540.54   834.5 2560.75  849.432571.789   853.3    2575
#Mann= 8 ,-1 , 0
       0      .1       0  441.09    .045       0  461.09     .06       0
  578.57      .1       0  605.97      .1       0     714      .1       0
  748.41      .1       0  849.43      .1       0
#XS Ineff= 2 , 0
          421.71 2488.92
Permanent Ineff=
       F       F
Bank Sta=441.09,461.09
XS Rating Curve= 0 ,0
Exp/Cntr(USF)=0,0
Exp/Cntr=0.3,0.1

Type RM Length L Ch R = 1 ,33627   ,243,238.7,234.2
XS GIS Cut Line= 3
2413468.80465614594770.2816805152413766.33565123594665.495782922
     2414101.112      594234.267
#Sta/Elev= 30
       0  2548.2    23.3 2547.74    38.9 2545.09    94.1 2540.87   174.6 2532.42
     217 2526.42   251.2 2518.63   284.9 2512.34   328.3 2489.46   339.4 2484.94
   379.3 2484.54     385 2482.76     391 2477.22  395.092475.962   405.2  2475.1
  413.882475.856   420.4 2479.27     425 2480.07   483.7  2478.5   510.8 2481.46
   526.8 2480.22  543.882480.615   561.9 2481.49   612.8 2481.05  685.982485.735
   721.6 2486.79   733.1 2489.51   809.8 2531.54   829.3 2544.19   861.4 2563.01
#Mann= 5 ,-1 , 0
       0      .1       0  395.09    .045       0  413.88      .1       0
  543.88     .06       0  685.98      .1       0
#XS Ineff= 3 ,-1
  424.85  511.21 2480.26  511.21  652.43 2482.63  652.43   861.4 2480.26
Permanent Ineff=
       F       F       F
Bank Sta=395.09,413.88
XS Rating Curve= 0 ,0
Exp/Cntr(USF)=0,0
Exp/Cntr=0.3,0.1

Type RM Length L Ch R = 1 ,33388   ,189.1,194.3,199.5
XS GIS Cut Line= 2
      2413913.98      595036.844      2414186.85      594260.071
#Sta/Elev= 30
       0 2550.54    39.1 2542.71   112.7 2524.25   161.4 2506.05  177.322501.368
  194.762498.184   236.7 2493.64   259.5 2493.24  287.982494.527   315.1 2495.42
   333.1 2494.66   337.4 2493.37   345.8 2488.57   371.3 2471.47   379.7 2468.96
   392.5 2467.85  402.472463.556   403.2 2463.34   417.9 2462.44   422.8  2463.3
   431.2 2467.54   437.5 2469.11   478.3 2470.09   494.2 2472.58  509.282472.829
  619.932474.016   638.3 2477.55   663.4 2490.26   762.6  2548.9   823.3 2582.59
#Mann= 9 ,-1 , 0
       0     .05       0  177.32      .1       0  194.76     .05       0
  287.98      .1       0  402.47     .05       0   403.2    .045       0
   422.8     .05       0  509.28     .06       0  619.93      .1       0
Bank Sta=403.2,422.8
XS Rating Curve= 0 ,0
Exp/Cntr(USF)=0,0
Exp/Cntr=0.5,0.3

Type RM Length L Ch R = 1 ,33194   ,78.2,77.9,78.8
XS GIS Cut Line= 2
2413967.74591185595066.3993732582414467.74591183 594408.06603993
#Sta/Elev= 30
       0 2539.27    70.2 2521.61     121  2498.6   145.5 2489.24   158.1 2485.86
   183.8 2481.41   226.6 2478.14   332.3 2477.27     338 2475.57   359.9 2464.57
   386.6 2462.55   400.8  2457.7  406.692457.011   419.5 2455.66  432.192456.788
   449.3 2462.56     482 2463.69   497.1 2466.71   520.7 2466.48   545.1 2461.78
  560.212463.135   604.6 2467.31   624.5 2475.43     652 2489.35   667.8  2501.6
   717.6 2534.08   743.3 2553.18   757.6 2557.84   771.8 2571.47   826.7 2610.39
#Mann= 4 ,-1 , 0
       0     .05       0  406.69    .045       0  432.19     .06       0
  560.21      .1       0
#XS Ineff= 2 , 0
                          501.69            2467
Permanent Ineff=
       F       F
Bank Sta=406.69,432.19
XS Rating Curve= 0 ,0
Exp/Cntr(USF)=0,0
Exp/Cntr=0.5,0.3

Type RM Length L Ch R = 1 ,33116   ,255.6,256.8,257.2
XS GIS Cut Line= 2
2414023.47507851595119.524373258 2414523.4750785 594461.19103993
#Sta/Elev= 30
       0 2528.93    56.4 2519.92    71.6 2513.93   136.3 2484.83   167.7 2477.47
   227.3 2472.69   307.6  2471.8   314.1 2470.02   337.8 2459.92   386.8  2460.4
  400.092454.073   413.2 2453.16  423.092453.929     436 2458.34   459.6 2460.75
   513.1 2461.26   533.6 2458.37  545.972458.951   604.4 2464.72   611.7 2467.29
   638.7 2480.34     658 2491.02   690.1 2511.65   704.2 2522.47   715.8 2529.55
   754.6 2560.31   764.3 2561.79   767.1 2563.26   778.5  2573.6   826.7 2609.15
#Mann= 4 ,-1 , 0
       0     .05       0  400.09    .045       0  423.09     .06       0
  545.97      .1       0
#XS Ineff= 2 , 0
          384.44 2461.24  467.87         2463.04
Permanent Ineff=
       F       F
Bank Sta=400.09,423.09
XS Rating Curve= 0 ,0
Exp/Cntr(USF)=0,0
Exp/Cntr=0.5,0.3

Type RM Length L Ch R = 1 ,32859   ,161.5,168.6,175.2
XS GIS Cut Line= 2
2414187.34345853595295.1061609692414710.78445853594661.256160969
#Sta/Elev= 30
       0 2514.28    31.9 2506.68    73.4 2489.12   104.5  2478.3   141.1    2468
     172 2461.61   223.2 2456.66   277.5 2456.51   328.6 2452.77   374.3  2452.6
  389.082450.709  424.222444.984   430.9 2443.93  442.322444.962   455.6 2445.59
   468.1 2449.84   512.1 2448.22  535.932452.637     590 2463.97   633.6 2468.52
   654.4 2474.89   666.7 2481.49     688 2495.69   716.6 2517.62   732.2 2520.68
   737.4 2523.31   751.9 2540.66     786 2563.93   813.6  2578.8     822  2580.9
#Mann= 5 ,-1 , 0
       0     .05       0  389.08     .06       0  424.22    .045       0
  442.32     .06       0  535.93      .1       0
#XS Ineff= 2 , 0
                          472.42         2450.56
Permanent Ineff=
       F       F
Bank Sta=424.22,442.32
XS Rating Curve= 0 ,0
Exp/Cntr(USF)=0,0
Exp/Cntr=0.3,0.1

Type RM Length L Ch R = 1 ,32690   ,184,184,182.2
XS GIS Cut Line= 4
2414226.83413414595351.3468902352414494.63594634 595118.39829511
2414594.12863508595077.5881536192414755.41394634594886.562834126
#Sta/Elev= 30
       0 2517.38    56.5 2510.59    74.4 2506.45    88.3 2500.23     130  2475.7
   152.7 2465.31   171.9 2459.56   204.9 2454.27   257.9 2449.56   284.4 2449.47
   342.7 2445.06   392.5  2445.3   409.8 2439.99  422.792439.241   427.1 2438.86
  440.672439.187   458.1 2448.15   464.1 2447.75  475.282443.928   498.6 2440.26
   537.9 2442.72   577.7 2441.41   586.2  2443.5   594.7 2449.62   600.4  2452.1
  623.962455.161     643 2459.26   659.8 2466.38   702.6 2493.14   712.5 2501.89
#Mann= 5 ,-1 , 0
       0     .05       0  422.79    .045       0  440.67     .05       0
  475.28     .06       0  623.96      .1       0
#XS Ineff= 2 , 0
                          459.08            2449
Permanent Ineff=
       F       F
Bank Sta=422.79,440.67
XS Rating Curve= 0 ,0
Exp/Cntr(USF)=0,0
Exp/Cntr=0.3,0.1

Type RM Length L Ch R = 1 ,32506   ,146.7,147.7,146.5
XS GIS Cut Line= 4
2414228.71886586595375.1423536712414535.93543416595303.085404875
2414663.44214727 595240.474907262414854.57930001595021.794163422
#Sta/Elev= 30
       0 2514.72    25.4 2511.92    66.5 2509.85    87.7 2506.41   103.5 2500.37
   144.5 2476.88   189.7 2462.31   218.5 2456.97   271.9 2452.99   288.3 2449.08
     344 2444.28   358.9 2439.72   379.6 2437.55   391.8 2433.43  398.622433.068
   409.7 2432.06  416.722433.144   428.6 2434.21   445.6 2439.47   454.6  2436.9
   468.9 2435.55  562.972433.404   585.1 2433.99     605 2437.71   644.6 2435.56
   661.1 2436.39   683.3 2441.95  691.94 2445.52   721.9 2463.83     748 2482.29
#Mann= 5 ,-1 , 0
       0     .05       0  398.62    .045       0  416.72     .05       0
  562.97     .06       0  691.94      .1       0
#XS Ineff= 2 , 0
                          444.64          2439.6
Permanent Ineff=
       F       F
Bank Sta=398.62,416.72
XS Rating Curve= 0 ,0
Exp/Cntr(USF)=0,0
Exp/Cntr=0.3,0.1

Type RM Length L Ch R = 1 ,32359   ,149.2,144.7,138.5
XS GIS Cut Line= 4
2414449.36467316595751.4058341262414660.82521708595404.075675609
2414854.05430579595306.3227438382414982.08686586      595146.119
#Sta/Elev= 30
       0 2508.19    66.7 2502.52    90.1 2498.52   141.6  2488.4   183.7 2475.19
   197.8 2471.81   239.4 2467.54   307.8 2455.39   369.3 2437.23   416.2 2431.46
  436.682427.542   447.6 2426.93  455.882427.636   464.8 2432.49   474.5  2433.8
   483.5 2430.81   491.6 2429.64   580.9 2426.76  627.032429.434   656.7 2427.56
   685.2 2427.12   699.8 2427.56   716.5  2429.7     731 2429.52   745.8 2427.53
  761.012429.317   773.4 2431.51   782.3 2435.23   802.2 2446.08   828.3 2462.29
#Mann= 5 ,-1 , 0
       0     .05       0  436.68    .045       0  455.88     .05       0
  627.03     .06       0  761.01      .1       0
#XS Ineff= 2 , 0
                          473.51            2434
Permanent Ineff=
       F       F
Bank Sta=436.68,455.88
XS Rating Curve= 0 ,0
Exp/Cntr(USF)=0,0
Exp/Cntr=0.3,0.1

Type RM Length L Ch R = 1 ,32214   ,165.1,162.8,159.5
XS GIS Cut Line= 2
2414463.48510977595844.5022707342415043.94229756595174.775324391
#Sta/Elev= 30
       0 2513.85   113.4 2505.76   203.9 2492.36   228.9 2484.25   277.8 2460.24
   302.2 2451.74   320.3 2443.71   332.7    2437   354.4 2428.68   363.3 2426.72
   399.8 2425.77   408.3    2423   419.6 2422.53  424.282421.027   431.4 2419.79
  442.582420.911   473.2 2427.85   485.4 2425.39   589.8 2423.52   623.8 2424.53
   657.8 2427.18  701.962425.753   754.1 2425.77   772.4 2426.86   796.7 2424.63
   810.9 2426.03   817.8 2427.68   833.5 2433.84   852.9 2443.53   886.3  2463.8
#Mann= 5 ,-1 , 0
       0     .05       0  424.28    .045       0  442.58     .05       0
  701.96     .06       0   852.9      .1       0
#XS Ineff= 2 , 0
          379.34  2429.1  472.38         2428.08
Permanent Ineff=
       F       F
Bank Sta=424.28,442.58
XS Rating Curve= 0 ,0
Exp/Cntr(USF)=0,0
Exp/Cntr=0.3,0.1

Type RM Length L Ch R = 1 ,32051   ,161.7,158.3,154.5
XS GIS Cut Line= 2
2414716.78943416 595905.46619025     2415095.858      595194.288
#Sta/Elev= 30
       0 2494.04    26.1 2495.41    48.8 2491.46    69.3 2486.55   120.3 2465.87
   171.3 2439.77   184.7 2435.53   205.4 2431.43   234.6 2423.78   266.3 2418.98
   302.6  2417.8  325.232418.453   343.4 2419.52   369.3 2418.33   379.6 2414.41
   393.2 2413.14   400.9 2414.25   411.3 2419.33   415.9 2420.16   426.4 2419.04
  447.182419.771  569.122421.073  714.852423.177   733.1 2423.93   741.1 2426.37
   755.8 2432.75   773.9 2442.06   783.6 2448.08     795 2455.88   805.9 2464.92
#Mann= 7 ,-1 , 0
       0     .05       0  325.23      .1       0   379.6    .045       0
   400.9      .1       0  447.18     .05       0  569.12     .06       0
  714.85      .1       0
#XS Ineff= 2 , 0
          348.27 2423.44  418.87         2423.19
Permanent Ineff=
       F       F
Bank Sta=379.6,400.9
XS Rating Curve= 0 ,0
Exp/Cntr(USF)=0,0
Exp/Cntr=0.3,0.1

Type RM Length L Ch R = 1 ,31893   ,175.2,170.6,165
XS GIS Cut Line= 3
     2414890.872      595991.1312415019.70191952595722.061943891
     2415158.714      595216.589
#Sta/Elev= 30
       0 2471.77    45.1 2467.21    58.4 2461.59    76.2 2458.06    93.9  2451.1
   191.5 2429.66   226.9 2412.83   312.6 2414.33   335.1 2411.62   354.7 2412.92
   389.2  2412.7     397 2411.17  401.582408.821   409.9 2407.22   422.4  2407.5
  426.982408.771   443.1 2415.36   504.3 2414.35  649.672417.103   671.2 2417.36
   687.8  2419.6   708.6 2419.16   733.5 2420.54   745.9 2421.77  756.612424.552
   784.1 2436.94   795.7 2443.81   808.1 2453.02   816.4 2454.43   822.6 2457.98
#Mann= 5 ,-1 , 0
       0     .05       0  401.58    .045       0  426.98     .05       0
  649.67     .06       0  756.61      .1       0
#XS Ineff= 2 , 0
          355.97 2417.42
Permanent Ineff=
       F       F
Bank Sta=401.58,426.98
XS Rating Curve= 0 ,0
Exp/Cntr(USF)=0,0
Exp/Cntr=0.3,0.1

Type RM Length L Ch R = 1 ,31722   ,138.1,134,131.3
XS GIS Cut Line= 3
2415102.47667806596039.1409731722415215.18505366595708.934836578
     2415201.664      595223.879
#Sta/Elev= 30
       0 2448.09    68.4  2446.9      98 2444.26   119.1 2437.84     136 2436.24
   186.7 2417.97   203.6 2415.13   220.5 2408.53   232.8 2405.95   258.6 2405.35
   283.9 2407.15   313.5 2404.99   334.6 2407.15   379.4 2407.86   387.4 2406.91
  403.082401.677   415.1 2400.57  427.082401.815   443.4  2406.2  590.812409.605
   647.5 2411.58   683.5 2416.34   739.5 2417.51   763.5 2424.63  787.432437.175
   795.5 2442.61   807.5 2445.29   811.5 2447.34   822.9 2457.32   834.2 2465.01
#Mann= 5 ,-1 , 0
       0     .05       0  403.08    .045       0  427.08     .05       0
  590.81     .06       0  787.43      .1       0
#XS Ineff= 2 , 0
          365.28 2410.36
Permanent Ineff=
       F       F
Bank Sta=403.08,427.08
XS Rating Curve= 0 ,0
Exp/Cntr(USF)=0,0
Exp/Cntr=0.3,0.1

Type RM Length L Ch R = 1 ,31588   ,151.2,152.6,150.1
XS GIS Cut Line= 3
 2415359.5735683596016.1826487812415355.45070244595665.127458531
     2415254.739      595216.017
#Sta/Elev= 30
       0 2415.73    41.8 2411.48   129.8 2409.64   177.6 2406.51   201.6 2404.51
   241.2 2399.07   265.8 2398.81   285.8 2400.85   333.8 2400.11   353.8 2401.68
     362 2403.55  375.222398.106   378.4 2397.46  403.022397.894   415.3 2400.25
   456.3 2402.81   509.6 2403.38   558.8  2405.7  569.782407.112   600.1 2411.72
   628.4 2412.39   637.1 2413.62  667.522413.879   685.8 2413.97   706.3 2417.46
   722.7 2426.91     735 2429.03   739.1 2430.72     776 2458.36   811.3 2482.64
#Mann= 5 ,-1 , 0
       0     .05       0  375.22    .045       0  403.02     .05       0
  569.78     .06       0  667.52      .1       0
#XS Ineff= 2 , 0
          360.77  2405.2
Permanent Ineff=
       F       F
Bank Sta=375.22,403.02
XS Rating Curve= 0 ,0
Exp/Cntr(USF)=0,0
Exp/Cntr=0.3,0.1

Type RM Length L Ch R = 1 ,31436   ,114.3,105,95.2
XS GIS Cut Line= 3
2415489.19565123596005.5040536562415508.55605366595649.718458532
      2415368.22       595195.28
#Sta/Elev= 30
       0 2409.06    31.1 2404.77    47.2 2404.37    75.2 2400.81   123.3 2396.97
   179.3 2396.73   215.4 2394.56   279.5 2393.57   295.5 2395.22   359.7 2396.03
     389 2397.99  401.612391.788   414.1 2390.91  419.112391.622   447.6 2395.94
  486.662396.662     569 2401.06   594.1  2405.7   656.9 2408.21  683.792412.886
   694.6 2414.06   715.5 2419.16   728.1 2425.38   736.5  2431.2     749 2444.45
   761.6 2453.78   770.9 2462.72   782.5 2476.02   798.4 2487.58   831.9 2508.83
#Mann= 5 ,-1 , 0
       0     .05       0  401.61    .045       0  419.11     .05       0
  486.66     .06       0  683.79      .1       0
#XS Ineff= 2 , 0
          385.57  2402.4
Permanent Ineff=
       F       F
Bank Sta=401.61,419.11
XS Rating Curve= 0 ,0
Exp/Cntr(USF)=0,0
Exp/Cntr=0.5,0.3

Type RM Length L Ch R = 1 ,31331   ,106.2,104.4,102.7
XS GIS Cut Line= 4
  2415657.179961595971.4443869942415655.91865492 595604.74572744
2415540.81448825 595514.120727442415445.50198828595175.058227425
#Sta/Elev= 30
       0 2400.55      45 2400.04      85 2395.69     133 2393.89     165 2389.18
     193 2387.55   271.9 2388.72     297 2387.95     309 2389.02   330.2  2388.1
  379.852389.923   415.7 2391.37   427.2  2395.1  434.222393.562   447.1 2388.64
   456.6 2387.85   469.9 2388.67   486.8 2393.24  513.112394.284   566.8 2395.82
   591.8 2401.42  611.372403.131     674 2408.24   703.9 2419.74   716.4 2429.08
   728.9 2430.69   737.2 2438.21   774.6 2461.65   845.2 2509.94   865.4 2524.89
#Mann= 7 ,-1 , 0
       0     .05       0  379.85     .06       0  434.22     .05       0
   447.1    .045       0   469.9     .05       0  513.11     .06       0
  611.37      .1       0
#XS Ineff= 2 , 0
          427.28 2395.68   527.5            2392
Permanent Ineff=
       F       F
Bank Sta=447.1,469.9
XS Rating Curve= 0 ,0
Exp/Cntr(USF)=0,0
Exp/Cntr=0.5,0.3

Type RM Length L Ch R = 1 ,31226   ,128.4,144.4,158.2
XS GIS Cut Line= 4
2415718.98551655595912.4166092162415717.72421047595545.717949662
 2415602.6200438595455.0929496622415507.30754383595116.030449647
#Sta/Elev= 30
       0 2396.62      54  2391.8      82 2387.78   270.7 2386.62  327.042387.613
   372.3 2389.56   378.4 2389.32   397.8 2385.41   410.7 2384.43   423.7 2385.05
   448.7 2391.34   481.9 2393.44   522.1 2398.67  562.172401.673   586.1 2404.01
   596.9 2406.52     622 2419.23   634.8 2427.75   646.8 2437.25   659.3 2439.95
   663.4 2442.26   675.9 2449.89   684.2 2457.46   721.6 2484.75   738.2 2492.05
   746.5 2498.52   767.3 2511.47   801.1 2534.78   842.1 2560.96   865.4 2577.69
#Mann= 5 ,-1 , 0
       0     .05       0  327.04     .06       0   397.8    .045       0
   423.7     .06       0  562.17      .1       0
#XS Ineff= 2 , 0
          375.42  2398.5
Permanent Ineff=
       F       F
Bank Sta=397.8,423.7
XS Rating Curve= 0 ,0
Exp/Cntr(USF)=0,0
Exp/Cntr=0.5,0.3

Type RM Length L Ch R = 1 ,31082   ,251.3,245.7,240.2
XS GIS Cut Line= 2
2415859.04365492595919.1554496452415787.51587712595099.711005198
#Sta/Elev= 30
       0 2391.84    36.9 2388.37     102 2387.99   129.2    2386   141.2  2382.3
   149.3 2381.51  254.542381.493   285.8 2383.42   323.6 2382.62   370.1 2384.48
  381.48 2379.93     390 2378.88  399.082380.149   410.2 2386.56   414.3 2387.13
   434.3 2388.44  450.042385.784   478.5 2388.31   495.9 2395.07   526.7 2414.18
     615 2475.15   619.1 2477.57   631.1 2480.34   639.1 2487.93   647.1 2493.52
   675.2 2506.58   699.3 2521.01   723.4  2529.3   735.4 2538.53   822.6 2580.53
#Mann= 5 ,-1 , 0
       0     .05       0  254.54     .06       0  381.48    .045       0
  399.08     .06       0  450.04      .1       0
#XS Ineff= 2 , 0
          361.89  2394.5
Permanent Ineff=
       F       F
Bank Sta=381.48,399.08
XS Rating Curve= 0 ,0
Exp/Cntr(USF)=0,0
Exp/Cntr=0.3,0.1

Type RM Length L Ch R = 1 ,30836   ,141.3,144.9,147.3
XS GIS Cut Line= 3
2416017.03173417595911.4482414542416065.30372927595487.080756094
     2415853.249      595090.137
#Sta/Elev= 30
       0 2391.68    37.3    2390    53.4 2387.93     150 2386.92     158 2387.78
   170.1 2385.97   190.2 2377.08   218.4 2375.15  280.582373.792   381.72373.364
   415.6 2373.02   442.4 2374.77  460.122370.737     469 2369.88  478.222370.874
   486.7  2377.2   504.9 2379.31   522.2 2384.02   527.6 2386.72   577.4 2417.77
     650 2465.39   677.2 2485.42   690.8 2487.78     718 2509.69   731.6 2513.76
   740.9 2521.75   763.3 2535.82   804.2 2557.43   831.4 2567.67   877.1  2589.3
#Mann= 5 ,-1 , 0
       0     .05       0  280.58    .055       0   381.7      .1       0
  460.12    .045       0  478.22      .1       0
#XS Ineff= 2 , 0
          443.07  2382.5
Permanent Ineff=
       F       F
Bank Sta=460.12,478.22
XS Rating Curve= 0 ,0
Exp/Cntr(USF)=0,0
Exp/Cntr=0.3,0.1

Type RM Length L Ch R = 1 ,30691   ,419.4,408.1,405.7
XS GIS Cut Line= 3
2416069.26068653595898.3563772652416204.62872927595488.207214625
      2416064.21      595006.897
#Sta/Elev= 30
       0 2388.74    45.8 2386.53    92.6 2388.06   146.9 2386.53   172.1 2382.35
   197.4 2373.99   235.1 2371.95   290.1 2372.15   353.3  2369.6   374.3 2370.88
   460.3 2369.65   473.2 2368.81   483.3 2364.94   504.82365.125   518.4 2363.51
   526.22364.775   554.1 2375.65   570.8  2391.9   583.3 2396.79   592.5 2405.08
   608.3 2415.21   708.7 2472.58   724.8 2482.85   737.5 2485.09     750  2494.3
     800 2521.33   811.9 2528.93     825 2532.81   840.9  2542.9   933.3 2589.36
#Mann= 6 ,-1 , 0
       0     .06       0  116.92      .1       0  257.63     .06       0
  384.92      .1       0   504.8    .045       0   526.2      .1       0
#XS Ineff= 2 , 0
          444.19    2380
Permanent Ineff=
       F       F
Bank Sta=504.8,526.2
XS Rating Curve= 0 ,0
Exp/Cntr(USF)=0,0
Exp/Cntr=0.3,0.1

Type RM Length L Ch R = 1 ,30283   ,194.2,191.9,190.4
XS GIS Cut Line= 2
     2416801.181      595605.7082416310.16213659594959.990512188
#Sta/Elev= 30
       0 2472.04  101.072422.601   112.4 2417.77   164.9 2389.23   169.9 2385.39
   179.9 2374.87   204.9 2372.91   230.2  2356.1   237.9 2352.93   244.9 2351.62
   264.9 2352.61   290.5  2350.8     304 2352.75  322.852353.043   345.8 2351.65
   370.5 2355.02   387.6 2349.63     396 2349.02   413.3 2349.57   431.2 2355.34
   484.7 2358.26   504.7 2363.68   568.3 2405.89   604.6 2427.32   627.7 2438.48
   677.4 2460.24     693 2463.22   707.5 2470.89   773.1 2496.83   811.2 2509.37
#Mann= 5 ,-1 , 0
       0      .1       0  101.07     .06       0  322.85      .1       0
   387.6    .045       0   413.3      .1       0
#XS Ineff= 2 , 0
          367.53 2359.08
Permanent Ineff=
       F       F
Bank Sta=387.6,413.3
XS Rating Curve= 0 ,0
Exp/Cntr(USF)=0,0
Exp/Cntr=0.3,0.1
